--- RASTutorial.prj (project) ---

Proj Title=RASTutorial
Current Plan=p01
Default Exp/Contr=0.3,0.1
English Units
Geom File=g01
Unsteady File=u01
Plan File=p01
Y Axis Title=Elevation
X Axis Title(PF)=Main Channel Distance
X Axis Title(XS)=Station
BEGIN DESCRIPTION:
END DESCRIPTION:
DSS File=dss
DSS Export Rating Curves= 0
DSS Export Rating Curve Sorted= 0
DSS Export Volume Flow Curves= 0
DXF OffsetX= 0
DXF OffsetY= 0
DXF ScaleX= 1
DXF ScaleY= 10

--- RASTutorial.p01 (plan) ---

Plan Title=Q50
Program Version=6.00
Short Identifier=Q50
Simulation Date=06JUL2021,0000,06JUL2021,0400
Geom File=g01
Flow File=u01
Subcritical Flow
K Sum by GR= 0
Std Step Tol= 0.01
Critical Tol= 0.01
Num of Std Step Trials= 20
Max Error Tol= 0.3
Flow Tol Ratio= 0.001
Split Flow NTrial= 30
Split Flow Tol= 0.02
Split Flow Ratio= 0.02
Log Output Level= 0
Friction Slope Method= 1
Unsteady Friction Slope Method= 2
Unsteady Bridges Friction Slope Method= 1
Parabolic Critical Depth
Global Vel Dist= 0 , 0 , 0
Global Log Level= 0
CheckData=True
Encroach Param=-1 ,0,0, 0
Computation Interval=5SEC
Output Interval=10MIN
Instantaneous Interval=10MIN
Mapping Interval=10MIN
Computation Time Step Use Courant=        0
Computation Time Step Use Time Series=    0
Computation Time Step Count To Double=0
Computation Time Step Max Doubling=0
Computation Time Step Max Halving=0
Computation Time Step Residence Courant=0
Computation Time Step TS=, 0
Computation Time Step TS=, 0
Computation Time Step TS=, 0
Computation Time Step TS=, 0
Computation Time Step TS=, 0
Computation Time Step TS=, 0
Computation Time Step TS=, 0
Computation Time Step TS=, 0
Computation Time Step TS=, 0
Computation Time Step TS=, 0
Computation Time Step TS=, 0
Computation Time Step TS=, 0
Computation Time Step TS=, 0
Computation Time Step TS=, 0
Computation Time Step TS=, 0
Computation Time Step TS=, 0
Computation Time Step TS=, 0
Computation Time Step TS=, 0
Computation Time Step TS=, 0
Computation Time Step TS=, 0
Computation Time Step TS=, 0
Computation Time Step TS=, 0
Computation Time Step TS=, 0
Computation Time Step TS=, 0
Computation Time Step TS=, 0
Computation Time Step TS=, 0
Computation Time Step TS=, 0
Computation Time Step TS=, 0
Computation Time Step TS=, 0
Computation Time Step TS=, 0
Computation Time Step TS=, 0
Computation Time Step TS=, 0
Computation Time Step TS=, 0
Computation Time Step TS=, 0
Computation Time Step TS=, 0
Computation Time Step TS=, 0
Computation Time Step TS=, 0
Computation Time Step TS=, 0
Computation Time Step TS=, 0
Computation Time Step TS=, 0
Computation Time Step TS=, 0
Computation Time Step TS=, 0
Computation Time Step TS=, 0
Computation Time Step TS=, 0
Computation Time Step TS=, 0
Computation Time Step TS=, 0
Computation Time Step TS=, 0
Computation Time Step TS=, 0
Computation Time Step TS=, 0
Computation Time Step TS=, 0
Run HTab=-1
Run UNet=-1
Run Sediment= 0
Run PostProcess=-1
Run WQNet= 0
Run RASMapper= 0
UNET Theta= 1
UNET Theta Warmup= 1
UNET ZTol= 0.02
UNET ZSATol= 0.02
UNET MxIter= 20
UNET Max Iter WO Improvement= 0
UNET MaxInSteps= 0
UNET DtIC= 0
UNET DtMin= 0
UNET MaxCRTS= 20
UNET WFStab= 2
UNET SFStab= 1
UNET WFX= 1
UNET SFX= 1
UNET Gravity=32.174
UNET 1D Methodology=Finite Difference
UNET DSS MLevel= 4
UNET Pardiso=0
UNET DZMax Abort= 100
UNET Use Existing IB Tables=-1
UNET Froude Reduction=False
UNET Froude Limit= 0.8
UNET Froude Power= 4
UNET D1 Cores= 0
UNET WindReference=Eulerian
UNET WindDragFormulation=Hsu (1988)
UNET D2 Coriolis=0
UNET D2 Cores= 0
UNET D2 Theta= 1
UNET D2 Theta Warmup= 1
UNET D2 Z Tol= 0.01
UNET D2 Volume Tol= 0.01
UNET D2 Max Iterations= 20
UNET D2 Equation= 0
UNET D2 RampUpFraction=0.1
UNET D2 TimeSlices= 1
UNET D2 Turbulence Formulation=None
UNET D2 Eddy Viscosity=0.3
UNET D2 Transverse Eddy Viscosity=0.1
UNET D2 Smagorinsky Mixing=0.05
UNET D2 BCVolumeCheck=0
UNET D2 Cores=0
UNET D2 SolverType=PARDISO (Direct)
UNET D2 Minimum Iterations= 0
UNET D2 Maximum Iterations= 0
UNET D2 Restart Number= 10
UNET D2 Relaxation Coeff=1.3
UNET D2 SOR Precondition Iterations= 10
UNET D2 ILUT Maximum Fill= 8
UNET D2 ILUT Tolerance=1E-08
UNET D2 Name=I-35 Voronoi
UNET D2 Theta= 1
UNET D2 Theta Warmup= 1
UNET D2 Z Tol= 0.01
UNET D2 Volume Tol= 0.01
UNET D2 Max Iterations= 20
UNET D2 Equation= 2
UNET D2 RampUpFraction=0.1
UNET D2 TimeSlices= 1
UNET D2 Turbulence Formulation=None
UNET D2 Eddy Viscosity=0.3
UNET D2 Transverse Eddy Viscosity=0.1
UNET D2 Smagorinsky Mixing=0.05
UNET D2 BCVolumeCheck=0
UNET D2 Cores=0
UNET D2 SolverType=PARDISO (Direct)
UNET D2 Minimum Iterations= 0
UNET D2 Maximum Iterations= 0
UNET D2 Restart Number= 10
UNET D2 Relaxation Coeff=1.3
UNET D2 SOR Precondition Iterations= 10
UNET D2 ILUT Maximum Fill= 0
UNET D2 ILUT Tolerance=0
UNET D1D2 MaxIter= 0
UNET D1D2 ZTol=0.01
UNET D1D2 QTol=0.1
UNET D1D2 MinQTol=1
DSS File=dss
Write IC File= 0
Write IC File at Fixed DateTime=0
Write IC File at Sim End=0
Echo Input=False
Echo Parameters=False
Echo Output=False
Write Detailed= 0
HDF Write Warmup=0
HDF Write Time Slices=0
HDF Flush=0
HDF Additional Output Variable=Cell Hydraulic Depth
HDF Additional Output Variable=Cell Invert Depth (WSE - Cell Min Elev)
HDF Additional Output Variable=Cell Velocity
HDF Compression= 1
HDF Chunk Size= 1
HDF Spatial Parts= 1
HDF Use Max Rows=0
HDF Fixed Rows= 1
Calibration Method= 0
Calibration Iterations= 20
Calibration Max Change=0.05
Calibration Tolerance=0.2
Calibration Maximum=1.5
Calibration Minimum=0.5
Calibration Optimization Method= 1
WQ AD Non Conservative
WQ ULTIMATE=-1
WQ Max Comp Step=1HOUR
WQ Output Interval=15MIN
WQ Output Selected Increments= 0
WQ Output face flow=0
WQ Output face velocity=0
WQ Output face area=0
WQ Output face dispersion=0
WQ Output cell volume=0
WQ Output cell surface area=0
WQ Output cell continuity=0
WQ Output cumulative cell continuity=0
WQ Output face conc=0
WQ Output face dconc_dx=0
WQ Output face courant=0
WQ Output face peclet=0
WQ Output face adv mass=0
WQ Output face disp mass=0
WQ Output cell mass=0
WQ Output cell source sink temp=0
WQ Output nsm pathways=0
WQ Output nsm derived pathways=0
WQ Create Restart=0
WQ Fixed Restart=0
WQ System Summary=0
WQ Write To DSS=0
Sorting and Armoring Iterations= 10
XS Update Threshold= 0.02
Bed Roughness Predictor= 0
Hydraulics Update Threshold= 0.02
Energy Slope Method= 1
Volume Change Method= 1
Sediment Retention Method= 0
Sediment TS Multiplier= 1
Warm Up Method= 0
XS Weighting Method= 0
Number of US Weighted Cross Sections= 1
Number of DS Weighted Cross Sections= 1
Upstream XS Weight=0
Main XS Weight=1
Downstream XS Weight=0
Number of DS XS's Weighted with US Boundary= 1
Upstream Boundary Weight= 1
Weight of XSs Associated with US Boundary= 0
Number of US XS's Weighted with DS Boundary= 1
Downstream Boundary Weight= 0.5
Weight of XSs Associated with DS Boundary= 0.5
Percentile Method= 0
Sediment Output Level= 3
Mass or Volume Output= 0
Output Increment Type= 1
Profile and TS Output Increment= 1
Transport Output Increment 1
XS Output Flag= 0
XS Output Increment= 10
Read HDF5 Sediment Hotstart= 0
Sediment Hotstart Type= 0
Write Gradation File= 0
Read Gradation Hotstart= 0
Write HDF5 File= 1
Write Binary Output= 1
Write DSS Sediment File= 0
DSS Sediment Output Type= 1
SV Curve= 0
Specific Gage Flag= 0
Subcell Erosion Methods= 0
Subcell Deposition Methods= 0
Advection Scheme= 1
Matrix Solver= 0
Implicit Weighting Factor= 1
Maximum Outer Loop Convergence Iterations= 5
Convergence Maximum Absolute= 0.001
Convergence RMSE= 0.0001
Grain Fractions Max Abs Error= 0.001
Max Subgrid Regions= 1
Max Subgrid Length Scale= 3.402823E+38
Initial Layer Thickness= 3.402823E+38
Min Layer Thickness= 3.402823E+38
Max Layer Thickness= 3.402823E+38
Number of Layers= 5

--- RASTutorial.u01 (unsteady flow) ---

Flow Title=Q50
Program Version=6.00
Use Restart= 0
Boundary Location=                ,                ,        ,        ,                ,I-35 Voronoi    ,                ,Upstream
Interval=4HOUR
Flow Hydrograph= 2
  178208  178208
Stage Hydrograph TW Check=0
Flow Hydrograph Slope= 0.001
Use DSS=False
Use Fixed Start Time=False
Is Critical Boundary=False
Boundary Location=                ,                ,        ,        ,                ,I-35 Voronoi    ,                ,Downstream
Interval=4HOUR
Stage Hydrograph= 2
     896     896
Stage Hydrograph Use Initial Stage=-1
Stage Hydrograph TW Check=0
Use DSS=False
Use Fixed Start Time=False
Is Critical Boundary=False
Precipitation Mode=Disable
Wind Mode=No Wind Forces
Met BC=Precipitation|Expanded View=0
Met BC=Precipitation|Point Interpolation=Nearest
Met BC=Precipitation|Gridded Source=DSS
Met BC=Evapotranspiration|Expanded View=0
Met BC=Evapotranspiration|Point Interpolation=Nearest
Met BC=Evapotranspiration|Gridded Source=DSS
Met BC=Wind Speed|Expanded View=0
Met BC=Wind Speed|Constant Units=ft/s
Met BC=Wind Speed|Point Interpolation=Nearest
Met BC=Wind Speed|Gridded Source=DSS
Met BC=Wind Direction|Expanded View=0
Met BC=Wind Direction|Point Interpolation=Nearest
Met BC=Wind Direction|Gridded Source=DSS
Met BC=Wind Velocity X|Expanded View=0
Met BC=Wind Velocity X|Constant Units=ft/s
Met BC=Wind Velocity X|Point Interpolation=Nearest
Met BC=Wind Velocity X|Gridded Source=DSS
Met BC=Wind Velocity Y|Expanded View=0
Met BC=Wind Velocity Y|Constant Units=ft/s
Met BC=Wind Velocity Y|Point Interpolation=Nearest
Met BC=Wind Velocity Y|Gridded Source=DSS
Met BC=Air Density|Mode=Constant
Met BC=Air Density|Expanded View=0
Met BC=Air Density|Constant Value=1.225
Met BC=Air Density|Point Interpolation=Nearest
Met BC=Air Density|Gridded Source=DSS
Met BC=Air Temperature|Expanded View=0
Met BC=Air Temperature|Point Interpolation=Nearest
Met BC=Air Temperature|Gridded Source=DSS
Met BC=Humidity|Expanded View=0
Met BC=Humidity|Point Interpolation=Nearest
Met BC=Humidity|Gridded Source=DSS
Met BC=Air Pressure|Expanded View=0
Met BC=Air Pressure|Point Interpolation=Nearest
Met BC=Air Pressure|Gridded Source=DSS
Non-Newtonian Method= 0 ,
Non-Newtonian Constant Vol Conc=0
Non-Newtonian Yield Method= 0 ,
Non-Newtonian Yield Coef=0, 0
User Yeild=   0
Non-Newtonian Sed Visc= 0 ,
Non-Newtonian Obrian B=0
User Viscosity=0
User Viscosity Ratio=0
Herschel-Bulkley Coef=0, 0
Clastic Method= 0 ,
Coulomb Phi=0
Voellmy X=0
Non-Newtonian Hindered FV= 0
Non-Newtonian FV K=0
Non-Newtonian ds=0
Non-Newtonian Max Cv=0
Non-Newtonian Bulking Method= 0 ,
Non-Newtonian High C Transport= 0 ,

--- RASTutorial.g01 (geometry) ---

Geom Title=Grid1
Program Version=6.00

Storage Area=I-35 Voronoi    ,,
Storage Area Surface Line= 6
2164465.29042785362589.954963321
2158337.41570331358260.236463966
        2154063.         358455.
2154537.00222513361382.668094223
        2162504.         364731.
2164465.29042785362589.954963321
Storage Area Type= 1
Storage Area Is2D=-1
Storage Area Point Generation Data=0,0,1500,1500
Storage Area 2D Points= 3843
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Storage Area Mannings=0.03
2D Cell Volume Filter Tolerance=0.01
2D Cell Minimum Area Fraction=0.01
2D Face Profile Filter Tolerance=0.01
2D Face Area Elevation Profile Filter Tolerance=0.01
2D Face Area Elevation Conveyance Ratio=0.02
2D Face Area Laminar Depth=0.2

BC Line Name=Upstream
BC Line Storage Area=I-35 Voronoi
BC Line Start Position= 2154744.62301645 , 357673.919636224
BC Line Middle Position= 2154369.74301645 , 358040.989636224
BC Line End Position= 2153994.86301645 , 358408.059636224
BC Line Arc= 2
2154744.62301645357673.9196362242153994.86301645358408.059636224

BC Line Name=Downstream
BC Line Storage Area=I-35 Voronoi
BC Line Start Position= 2164514.15770734 , 362627.627183707
BC Line Middle Position= 2163526.32580536 , 363686.018507257
BC Line End Position= 2162538.49390338 , 364744.409830807
BC Line Arc= 2
2164514.15770734362627.6271837072162538.49390338364744.409830807
LCMann Table=0

Chan Stop Cuts=-1
Use User Specified Reach Order=0
Composite Channel Slope=5
