--- RASTutorial.prj (project) ---

Proj Title=RASTutorial
Current Geom=g01
FOOT
Geom File=g01

--- RASTutorial.g01 (geometry) ---

Geom Title=Grid1
Program Version=5.00

Storage Area=I-35 Voronoi, 2159269.5, 361225.45012367493
Storage Area Surface Line= 6
2164465.29042785362589.954963321
2158337.41570331358260.236463966
       2154063.0        358455.0
2154537.00222513361382.668094223
       2162504.0        364731.0
2164465.29042785362589.954963321
Storage Area Type= 0
Storage Area Is2D=-1
Storage Area Point Generation Data=0,0,1500,1500
Storage Area 2D Points= 3843
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Storage Area Mannings=0.03
2D Cell Volume Filter Tolerance=0.01
2D Face Profile Filter Tolerance=0.01
2D Face Area Elevation Profile Filter Tolerance=0.01
2D Face Area Elevation Conveyance Ratio=0.02
LCMann Table=0

Chan Stop Cuts=-1
Use User Specified Reach Order=0
Composite Channel Slope=5
